--- E122-00-00.prj (project) ---

Proj Title=E122-00-00
Current Plan=p06
Default Exp/Contr=.3,.1
English Units
Geom File=g08
Flow File=f04
Flow File=f05
Plan File=p06
Plan File=p02
Y Axis Title=Elevation
X Axis Title(PF)=Main Channel Distance
X Axis Title(XS)=Station
BEGIN DESCRIPTION:
Watershed: White Oak Bayou
Stream Name: unnamed tributary to White Oak Bayou
HCFCD Unit E122-00-00
(Flood Hazard, Floodway) Model
10, 2, 1, .02% Event
File Name: E122-00-00.prj
Prepared by:  Ty Turner, Sean Sutton (TCB revisions) 6/10/03
Reviewed by: Joe Barrow
Status: Final RAS
END DESCRIPTION:
DSS Export Rating Curves= 0
DSS Export Rating Curve Sorted= 0
DSS Export Volume Flow Curves= 0
DXF OffsetX= 0
DXF OffsetY= 0
DXF ScaleX= 1
DXF ScaleY= 10

--- E122-00-00.p06 (plan) ---

Plan Title=FEMA Effective June 2007
Version=Version 3.0.1  Mar 2001
Short Identifier=FEMAeff0607
Geom File=g08
Flow File=f04
Subcritical Flow
K Sum by GR= 0
Std Step Tol= 0.01
Critical Tol= 0.01
Num of Std Step Trials= 20
Max Error Tol= 0.3
Flow Tol Ratio= 0.001
Split Flow NTrial= 30
Split Flow Tol= 0.02
Split Flow Ratio= 0.02
Log Output Level= 0
Friction Slope Method= 0
Unsteady Friction Slope Method= 2
Secant Critical Depth
Global Vel Dist= 0 , 0 , 0
Global Log Level= 0
CheckData=True
Encroach Param=-1 ,0,0, 2
Computation Interval=1HOUR
Output Interval=1HOUR
Run HTab= 0
Run UNet= 0
Run PostProcess= 0
UNET Theta= 1
UNET ZTol= 0.02
UNET ZSATol= 0.1
UNET MxIter= 20
UNET MaxInSteps= 20
UNET DtIC= 0
UNET DtMin= 0
UNET MaxCRTS= 20
UNET WFStab= 2
UNET SFStab= 1
UNET WFX= 1
UNET SFX= 1
UNET Convert EG Bridges=-1
UNET Use Existing IB Tables=-1
Instantaneous Interval=1HOUR
DSS File=dss
Write IC File= 0
IC Time=0
Write Velocity= 0
Write Detailed= 0

--- E122-00-00.p02 (plan) ---

Plan Title=Floodway
Version=Version 3.0.1  Mar 2001
Short Identifier=Floodway0607
Geom File=g08
Flow File=f05
Subcritical Flow
K Sum by GR= 0
Std Step Tol= 0.01
Critical Tol= 0.01
Num of Std Step Trials= 20
Max Error Tol= 0.3
Flow Tol Ratio= 0.001
Split Flow NTrial= 30
Split Flow Tol= 0.02
Split Flow Ratio= 0.02
Log Output Level= 0
Friction Slope Method= 0
Unsteady Friction Slope Method= 2
Secant Critical Depth
Global Vel Dist= 0 , 0 , 0
Global Log Level= 0
CheckData=True
Encroach Param=-1 ,0,0, 2
Encroach River=E122-00-00
Encroach Reach=E122-00-00_0000
Encroach Node=15316.87
       1 3611.96 3635.93
Encroach Node=15244.78
       1 3597.09 3679.09
Encroach Node=14980.69
       1 3624.54 3709.56
Encroach Node=14583.03
       1 3675.09 3756.53
Encroach Node=13856.36
       1 3821.34 3944.64
Encroach Node=13799.94
       1 3852.72 4002.43
Encroach Node=13754.94
       1 3923.52 4080.97
Encroach Node=13706.71
       1 3923.52 4080.97
Encroach Node=13661.82
       1 3965.62 4095.77
Encroach Node=13141.24
       1 4127.37 4229.76
Encroach Node=12779.21
       1 4045.27 4148.38
Encroach Node=11773.19
       1 3255.75 3356.98
Encroach Node=10772.07
       1 2443.73  2548.2
Encroach Node=9776.243
       1 1688.05 1792.28
Encroach Node=9412.584
       1 1291.29 1402.31
Encroach Node=9043.720
       1  821.61  930.76
Encroach Node=8817.703
       1  936.32 1055.41
Encroach Node=8751.316
       1  954.58 1068.79
Encroach Node=8747.55
       1  989.33 1120.14
Encroach Node=8706.955
       1  989.33 1120.14
Encroach Node=8630.772
       1 1036.09 1145.34
Encroach Node=8090.234
       1  1240.4 1354.92
Encroach Node=7366.673
       1 1652.34 1741.61
Encroach Node=7323.165
       1 1695.64 1780.64
Encroach Node=7296.664
       1 1107.64 2233.64
Encroach Node=7268.812
       1 1715.38 1809.38
Encroach Node=7249.799
       1 1728.43 1848.44
Encroach Node=6898.815
       1 1865.74 1949.85
Encroach Node=5983.005
       1 2265.55 2347.31
Encroach Node=5431.968
       1 2267.87 2341.36
Encroach Node=5380
       4       1
Encroach Node=5348.006
       1 2403.54 2499.54
Encroach Node=5267.653
       1 2397.92 2492.92
Encroach Node=4762.511
       1 2362.61 2470.62
Encroach Node=4689.561
       1  2359.4 2465.53
Encroach Node=4668.847
       1 2326.63 2467.86
Encroach Node=4648.134
       1 2326.63 2467.86
Encroach Node=4575.253
       1 2326.56 2483.56
Encroach Node=4230.466
       1 2329.89 2435.96
Encroach Node=3860.318
       1 2314.37 2423.06
Encroach Node=3809.425
       1 2299.79 2406.11
Encroach Node=3766.214
       1 2259.38 2409.28
Encroach Node=3049.070
       1  1626.4 1723.47
Encroach Node=2998.224
       1 1609.95 1710.26
Encroach Node=2111.142
       1 1391.51 1504.87
Encroach Node=2063.198
       1 1383.51 1498.45
Encroach Node=1748.955
       1 1286.99  1395.2
Encroach Node=1040.148
       1  883.52  987.78
Encroach Node=645.763
       1  520.08  616.15
Encroach Node=514.233
       1  257.29  335.35
Encroach Node=471.314
       1  212.29  327.92
Encroach Node=423.395
       1  212.29  327.92
Encroach Node=279.778
       1  163.39  268.64
Encroach Node=3.533
       1   89.99  192.71
Computation Interval=1HOUR
Output Interval=1HOUR
Run HTab= 0
Run UNet= 0
Run PostProcess= 0
UNET Theta= 1
UNET ZTol= 0.02
UNET ZSATol= 0.1
UNET MxIter= 20
UNET MaxInSteps= 20
UNET DtIC= 0
UNET DtMin= 0
UNET MaxCRTS= 20
UNET WFStab= 2
UNET SFStab= 1
UNET WFX= 1
UNET SFX= 1
UNET Convert EG Bridges=-1
UNET Use Existing IB Tables=-1
Instantaneous Interval=1HOUR
DSS File=dss
Write IC File= 0
IC Time=0
Write Velocity= 0
Write Detailed= 0

--- E122-00-00.f04 (steady flow) ---

Flow Title=FEMA Effective June 2007
Program Version=3.13
Number of Profiles= 4
Profile Names=10PCT_10yr,2PCT_50yr,1PCT_100yr,0.2PCT_500yr
River Rch & RM=E122-00-00,E122-00-00_0000            ,15316.87
    1212    1783    2072    2893
River Rch & RM=E122-00-00,E122-00-00_0000            ,14583.03
    1284    1890    2198    3072
River Rch & RM=E122-00-00,E122-00-00_0000            ,13799.94
    1355    1997    2323    3251
River Rch & RM=E122-00-00,E122-00-00_0000            ,12779.21
    1422    2099    2443    3423
River Rch & RM=E122-00-00,E122-00-00_0000            ,10772.07
    1496    2210    2573    3610
River Rch & RM=E122-00-00,E122-00-00_0000            ,8751.316
    1569    2322    2704    3798
River Rch & RM=E122-00-00,E122-00-00_0000            ,7366.673
    1653    2449    2853    4015
River Rch & RM=E122-00-00,E122-00-00_0000            ,5983.005
    1744    2588    3017    4252
River Rch & RM=E122-00-00,E122-00-00_0000            ,4689.561
    1830    2719    3172    4477
River Rch & RM=E122-00-00,E122-00-00_0000            ,3049.070
    1926    2868    3347    4733
River Rch & RM=E122-00-00,E122-00-00_0000            ,1040.148
    2023    3018    3525    4993
Boundary for River Rch & Prof#=E122-00-00,E122-00-00_0000            , 1
Up Type= 0
Dn Type= 3
Dn Slope=0.0012
DSS Import GetInterval= 0
DSS Import GetPeak= 0
DSS Import FillOption= 0
DSS File=V:\TSARP\4-EngCal\HydrologicModels\Klotz\E100_100_02\E100_100_02.dss

--- E122-00-00.f05 (steady flow) ---

Flow Title=Floodway
Program Version=3.13
Number of Profiles= 2
Profile Names=1PCT_100yr,1PCTFloodway_100yrFW
River Rch & RM=E122-00-00,E122-00-00_0000            ,15316.87
    2072    2072
River Rch & RM=E122-00-00,E122-00-00_0000            ,14583.03
    2198    2198
River Rch & RM=E122-00-00,E122-00-00_0000            ,13799.94
    2323    2323
River Rch & RM=E122-00-00,E122-00-00_0000            ,12779.21
    2443    2443
River Rch & RM=E122-00-00,E122-00-00_0000            ,10772.07
    2573    2573
River Rch & RM=E122-00-00,E122-00-00_0000            ,8751.316
    2704    2704
River Rch & RM=E122-00-00,E122-00-00_0000            ,7366.673
    2853    2853
River Rch & RM=E122-00-00,E122-00-00_0000            ,5983.005
    3017    3017
River Rch & RM=E122-00-00,E122-00-00_0000            ,4689.561
    3172    3172
River Rch & RM=E122-00-00,E122-00-00_0000            ,3049.070
    3347    3347
River Rch & RM=E122-00-00,E122-00-00_0000            ,1040.148
    3525    3525
Boundary for River Rch & Prof#=E122-00-00,E122-00-00_0000            , 1
Up Type= 0
Dn Type= 3
Dn Slope=0.0012
DSS Import GetInterval= 0
DSS Import GetPeak= 0
DSS Import FillOption= 0
DSS File=V:\TSARP\4-EngCal\HydrologicModels\Klotz\E100_100_02\E100_100_02.dss

--- E122-00-00.g08 (geometry) ---

Geom Title=E122-00-00 June 2007
Program Version=3.13

River Reach=E122-00-00      ,E122-00-00_0000
Reach XY= 30
     3071939.998    13896538.211     3072033.296    13894278.999
      3072052.64    13893084.268     3072087.297    13892418.796
     3072131.974    13892160.224     3072098.043    13891745.265
     3072145.865    13891531.949     3072204.164    13891474.993
     3072403.134    13891437.132     3073405.859    13891496.449
     3075827.853    13891571.174     3075940.153    13891514.218
     3075976.959    13891462.097     3076028.004    13890856.269
     3076087.647    13890668.475     3076117.737    13889507.595
     3076161.783    13889207.721     3076193.768    13888231.459
     3076339.382    13887908.261     3076400.853    13886243.048
     3076507.831    13886016.087     3076770.581    13885833.936
     3076850.105    13885691.546     3076882.612    13884863.804
     3076920.575    13884601.968     3077174.109    13884343.409
      3077707.13    13883884.806     3077786.923    13883718.774
     3077945.432    13883586.862     3077976.925    13883039.714

Type RM Length L Ch R = 1 ,15316.87,72.49,72.06,71.11
BEGIN DESCRIPTION:
E122-00-S5 (Survey 3611.96 to 3635.93) XS 2
Data inserted from bridge survey
Point deleted 149.94
END DESCRIPTION:
XS GIS Cut Line= 6
 3075675.648655713893830.6680771     3074690.159    13893723.694
     3072181.863    13893755.295     3072081.871    13893756.568
        3071891.       13893759.      3069935.56     13893783.91
#Sta/Elev= 30
  -30.71  106.01   14.74  102.23   44.92   104.6  224.53  102.46  501.37  104.51
  801.59  101.57 1181.86  104.88  1933.8   104.9 2030.35  102.27  2129.5  105.06
 2300.37     102 2401.97  105.01 2566.48  101.84 2613.59  104.66 2699.26  105.19
 2834.67  102.66 3003.11  105.59 3095.43  102.41 3258.63  105.67 3365.45   103.1
 3486.49  105.42 3611.96  105.19 3611.97   94.02 3635.87   94.02 3635.93  105.16
 3715.11  105.41 3842.72  103.28 4321.51  105.54  4724.2  104.37 5715.55  109.39
#Mann= 3 ,-1 , 0
  -30.71     .08       0 3486.49     .04       0 3715.11     .08       0
#XS Ineff= 2 , 0
         3559.96  106.19 3692.64          106.19
Permanent Ineff=
       F       F
Bank Sta=3611.96,3635.93
Exp/Cntr=0.5,0.3

Type RM Length L Ch R = 1 ,15244.78,262.96,264.1,265.65
BEGIN DESCRIPTION:
E122-00-SV5 (Survey 3585.09 to 3707.09) XS 1
END DESCRIPTION:
XS GIS Cut Line= 5
  3075692.20615813893793.1128294     3075667.331    13893790.333
     3074741.802    13893686.904     3072211.971    13893686.528
     3069945.965    13893686.528
#Sta/Elev= 30
  -25.03  106.25   17.79  102.17   67.28  104.62  240.34  102.31  560.23  104.97
  814.99  101.81 1702.64  105.17 2052.63  102.56 2172.63  105.12 2322.63  102.25
 2459.31  105.14 2577.63   101.9 2977.67  105.65 3127.71  101.99 3226.25  105.35
 3402.63  102.98 3550.82  106.29 3597.09  106.99 3632.09   92.53 3679.09  105.24
 3722.63  105.55 3867.63  103.13 4049.36  106.69 4197.63   104.5 4285.89  107.14
 4692.63  106.61 4739.36  104.46  4946.1  106.92 5027.84  104.49 5727.13  108.27
#Mann= 3 ,-1 , 0
  -25.03     .08       0 3550.82     .04       0 3722.63     .08       0
#XS Ineff= 2 , 0
         3584.74     108 3726.19          105.59
Permanent Ineff=
       F       F
Bank Sta=3597.09,3679.09
Exp/Cntr=0.3,0.1

Type RM Length L Ch R = 1 ,14980.69,390.82,397.66,403.94
BEGIN DESCRIPTION:
E122-00-V6 (Survey 3558.51 to 3709.56)
END DESCRIPTION:
XS GIS Cut Line= 6
 3075699.013712913893779.8662546     3074971.134    13893508.359
     3072261.131    13893428.957     3071982.309    13893420.836
     3071882.351    13893417.925     3069945.831    13893361.521
#Sta/Elev= 30
   -36.7  106.23    3.47  102.13  376.54  104.72 1010.95  101.74 1226.77  104.16
 1326.09  101.61 1486.05  104.69 2076.41  102.69 3034.44  105.41 3152.88  102.51
 3289.29  105.76 3411.98  103.47 3575.92  105.53 3624.54  107.56 3668.55   90.75
 3709.56  104.56 3748.95  105.33 3892.19     103 4030.46  105.96 4207.32     104
 4434.14  106.82 4505.33  103.93 4642.51  106.47 4786.24  102.85  4955.8  106.61
 5062.68  103.07  5107.7   105.7 5452.85  106.99 5587.91  103.36 5767.62  107.61
#Mann= 3 ,-1 , 0
   -36.7     .08       0 3575.92     .04       0 3748.95     .08       0
#XS Ineff= 2 , 0
          3614.7  107.65 3744.02          105.33
Permanent Ineff=
       F       F
Bank Sta=3624.54,3709.56
Exp/Cntr=0.3,0.1

Type RM Length L Ch R = 1 ,14583.03,732.35,726.67,717.31
BEGIN DESCRIPTION:
E122-00-SV6 (Survey 3663.06 to 3764.59) Pipeline location
END DESCRIPTION:
XS GIS Cut Line= 6
  3075705.477327 13893754.858261     3074889.887    13893397.909
     3072220.401    13893048.774     3072121.233    13893035.902
     3071901.664      13893007.4     3069986.569    13892758.806
#Sta/Elev= 30
  -31.13  106.19       0  102.34   343.3  104.86   992.3  101.29 1140.75   104.3
 1295.04  101.94 1695.98  104.93 1850.74  102.02 2034.44   104.9 2124.26  102.24
 2243.73   104.5 2654.57  102.06 2800.84   105.3 2986.67  101.66 3598.45  106.22
 3675.09  107.15 3717.97 89.8253 3724.95 93.9222 3752.37 99.9283 3756.53  104.63
 3772.56  104.19 4087.29   105.9 4272.31  103.11 4453.82  106.52 5119.35  103.36
 5318.82  105.73 5374.94  103.29 5500.48  107.08 5634.92  104.01 5803.94  106.76
#Mann= 3 ,-1 , 0
  -31.13     .08       0 3598.45     .04       0 3772.56     .08       0
#XS Ineff= 2 , 0
         3674.54  107.16 3831.99          106.19
Permanent Ineff=
       F       F
Bank Sta=3675.09,3756.53
Exp/Cntr=0.3,0.1

Type RM Length L Ch R = 1 ,13856.36,52.79,56.42,60.96
BEGIN DESCRIPTION:
E122-00-SV7 (Survey 3814.35 to 3944.64) XS 4
END DESCRIPTION:
XS GIS Cut Line= 6
 3075713.734643213893735.0764969        3073869.    13892778.117
     3072283.034    13892297.882     3072027.459    13892311.183
     3071927.594     13892316.38      3069994.81    13892318.044
#Sta/Elev= 30
  -31.01  106.21       0  102.59  355.74  104.67  986.39  101.19  1117.8  104.05
 1270.47  101.46 1447.61  104.02 1525.41  101.04 1624.69  104.86 1798.61  101.75
 2185.79  105.11 2341.38  101.31 2483.18  105.35 2613.62  101.68 2739.02  105.45
 2899.47  101.82 3130.87  105.29 3639.02  102.07 3775.56   105.2 3821.34   105.6
 3830.77   96.42 3855.07   90.76 3909.79   94.98 3944.64  104.75 4010.24  104.55
  4722.3  102.39  4842.3  105.34 5304.44  103.08 5453.85  106.31 5992.95  106.24
#Mann= 3 ,-1 , 0
  -31.01     .08       0 3775.56     .04       0 4010.24     .08       0
#XS Ineff= 2 , 0
         3814.19  106.21  3944.6          104.75
Permanent Ineff=
       F       F
Bank Sta=3821.34,3944.64
Exp/Cntr=0.5,0.3

Type RM Length L Ch R = 1 ,13799.94,91.4,93.23,90.8
BEGIN DESCRIPTION:
E122-00-S7 (Survey 3855.7 to 3946.89) XS 3
END DESCRIPTION:
XS GIS Cut Line= 6
 3075722.028194813893720.1422122     3073728.962    13892643.951
     3072488.338    13892259.721     3072182.591     13892252.14
     3071958.854    13892246.593     3070003.063    13892214.881
#Sta/Elev= 30
  -19.41  106.24    1.41  102.49  375.54  104.57  994.72  101.29 1110.29  103.47
  1524.7  101.22 1716.49  104.13 1806.81   101.9 2278.14  104.06    2345  101.14
 2516.26  104.62 2636.09  101.34 2762.08  105.26 2909.29  101.48 3045.07  104.83
 3427.03  101.84 3798.97  103.89 3852.72  104.49 3897.86   92.38  3921.9   89.95
 3957.41   94.22 4002.43  104.31 4768.95  102.23 4913.06  104.87 5067.58  102.75
 5260.73  105.31 5337.61  102.81  5416.2  105.54 5937.69  103.25 6030.11  105.38
#Mann= 3 ,-1 , 0
  -19.41     .08       0 3798.97     .04       0 4002.43     .08       0
#XS Ineff= 2 , 0
         3851.42   104.5 4002.58           104.5
Permanent Ineff=
       F       F
Bank Sta=3852.72,4002.43
Exp/Cntr=0.5,0.3

Type RM Length L Ch R = 3 ,13754.94,,,
BEGIN DESCRIPTION:
Structure 7 and 8 - West Road
END DESCRIPTION:
Bridge Culvert--1,0,-1,-1, 0
Deck Dist Width WeirC Skew NumUp NumDn MinLoCord MaxHiCord MaxSubmerge Is_Ogee
0.5,91,2.6,0, 86, 76, , , 0.95, 0, 0,0,,
     -20       0   29.86  177.38  348.32  400.86  599.73  696.53  704.54  748.98
   752.6  869.11 1019.97 1216.47 1288.71 1484.72 1543.95 1594.26 1714.66 1851.19
 2014.14 2123.73 2290.23 2307.65 2360.11 2379.97 2440.68 2528.92 2568.73 2584.18
 2623.08 2639.67 2657.01 2729.96 2746.24 2783.06 2835.62 2857.52 2898.24 2916.17
 2984.77 3333.17  3374.3 3403.95 3417.31  3437.8 3473.71 3775.88 3850.25 3861.29
 3901.32 3941.36 3981.37 4089.27 4224.17 4450.14  4496.9 4724.27 4776.85 4823.37
 4954.28 5005.13 5005.22 5022.86 5053.63 5074.84 5139.79 5156.07 5185.25 5219.46
 5289.39 5314.18 5325.82 5348.24 5373.93  5560.6 5582.37  5602.2 5631.05 5778.02
 5842.99 5879.17 5903.65 5940.47  5971.3    6031
     104     104     104     104     104     104     103     102     102     102
     102     102     102     102     102     102     102     103     103     103
     103     103     103     102     102     103     104     104     103     102
     102     103     104     105     105     104     103     102     102     103
     104     104     103     102     102     103     103     103  103.83   103.9
  104.06  104.05  103.93  103.61     103     103     103     103     103     104
     104     104     104     103     103     104     105     105     105     105
     104     103     103     104     105     105     104     104     105     105
     104     104     104     104     105     105
                                                                                
                                                                                
                                                                                
                                                                                
                                                                  101.43   101.5
  101.66  101.65  101.53  101.21
                                                                                
                                                                                
                                                
     -45       0   95.62  230.84  247.94  270.95  282.51  300.76  420.91  549.44
  647.09  925.62 1566.34 1666.92 1735.59 1925.92 2059.22 2086.97 2112.33 2216.32
 2254.74 2366.45 2452.64 2464.81 2511.67 2549.12 2566.07 2591.26 2619.48 2640.01
  2703.3  2745.4 2771.52  2825.9  2851.5 3105.81 3286.01 3311.74  3725.9 3788.09
 3794.56 3798.14 3801.72  3805.3 3808.87 3812.38 3815.79  3819.2 3822.61  3829.4
 3841.49 3852.15 3863.99 3869.57 3936.62  4056.7 4125.76 4209.27  4629.2 4631.24
 4731.48 4957.13  5088.6 5147.41 5153.92 5188.51 5428.47 5456.23  5497.2 5566.81
 5588.48 5714.63 5749.57 5810.25 5935.85    6102
     104     104     104     104     104     104     104     104     104     103
     102     102     103     103     103     103     103     103     103     103
     102     102     103     103     102     102     103     104     104     104
     104     103     102     102     103     103     103     103     103     103
     102     101     100      99      98      97      96      95      94      93
      92      92      93  103.02   103.7   103.7  103.37     103     103     103
     104     104     104     104     104     104     104     104     104     104
     104     104     104     104     104     104
                                                                                
                                                                                
                                                                                
                                                                                
                                                                                
                          100.72   101.4   101.4  101.07
                                                                                
                                                
Pier Skew, UpSta & Num, DnSta & Num=  ,3902.03, 4 ,3977.32, 4 , 3 , 3 , 0 ,,
     1.5     1.5       2       2
 89.9485   99.75   99.75  101.75
    1.35    1.35       2       2
 90.0842  100.11  100.11  102.11
Pier Skew, UpSta & Num, DnSta & Num=  ,3942.04, 4 ,4016.34, 4 , 3 , 3 , 0 ,,
     1.5     1.5       2       2
 89.9485   99.69   99.69  101.69
    1.35    1.35       2       2
 90.0842  100.15  100.15  102.15
BR Coef=-1 , 1 , 1 ,1.25, 0 ,,,0.8,-1,2,0,
WSPro=,,,, 1 ,,,, 0 ,,,, 0 ,,,,-1 ,-1 ,-1 , 0 , 0 , 0 , 0 , 0
BC Design=,, 0 ,, 0 ,,,,,,
BC HTab HWMax=106.24

Type RM Length L Ch R = 1 ,13706.71,48.18,44.89,41.12
BEGIN DESCRIPTION:
E122-00-S8 (Survey 3935.67 to 4045.74) XS 2
END DESCRIPTION:
XS GIS Cut Line= 6
  3075890.83385513893446.4657934     3073149.188    13892216.988
     3072985.617    13892203.726     3072536.715    13892170.277
      3071937.24    13892155.236     3070011.316    13892082.833
#Sta/Elev= 30
   -44.4  105.88       0  102.63  142.32  103.72  206.06  101.46  843.38  104.54
 1280.73  100.96  1408.3  104.71 1529.16  100.77 1598.18  103.89 1736.76  104.46
 1822.85  101.52 1967.07  104.75  2068.9  101.36 2219.32  104.14 2361.71   101.1
 2528.18     104  2608.2  101.42  2831.7  103.44 2885.42  100.99 2991.39  103.55
 3251.26  101.36 3904.96  104.07 3923.52  104.41 3960.69   92.39 3979.05   90.08
 4013.72    92.2 4039.74  100.64 4080.97  103.87 4088.01  103.85  6101.5  104.08
#Mann= 3 ,-1 , 0
   -44.4     .08       0 3904.96     .04       0 4088.01     .08       0
#XS Ineff= 2 , 0
          3923.2  104.42 4084.84          104.11
Permanent Ineff=
       F       F
Bank Sta=3923.52,4080.97
Exp/Cntr=0.5,0.3

Type RM Length L Ch R = 1 ,13661.82,504.11,520.58,519.26
BEGIN DESCRIPTION:
E122-00-SV8 (Survey 3938.67 to 4115.72) XS 1
END DESCRIPTION:
XS GIS Cut Line= 6
 3075900.701224713893383.9902531     3073149.188    13892146.255
     3072601.643     13892103.97     3072216.743    13892113.217
     3071924.015    13892120.249     3070011.316    13892049.821
#Sta/Elev= 30
  -21.31  105.82    2.29  102.21  986.79  101.65 1119.84  104.25 1260.94  100.95
 1391.69  104.45 1541.49  100.51 1686.82  104.58 1802.48  101.37 2002.03  104.59
 2080.19  101.36 2211.22  104.39 2347.43   101.3 2537.25  104.48 2613.97  101.15
 3058.55  104.36 3275.33  100.75 3425.27   104.6 3540.25  101.64 3615.02  104.68
 3816.21  101.99 3927.53  104.66 3965.62  105.89 4017.68   89.16 4056.81   92.25
 4095.77  105.16 4115.72   104.8 4266.35  102.11 4415.26  105.01 6136.77  104.72
#Mann= 3 ,-1 , 0
  -21.31     .08       0 3927.53     .04       0 4115.72     .08       0
#XS Ineff= 2 , 0
          3964.4  105.89 4095.57          105.16
Permanent Ineff=
       F       F
Bank Sta=3965.62,4095.77
Exp/Cntr=0.3,0.1

Type RM Length L Ch R = 1 ,13141.24,238.64,362.03,450.11
BEGIN DESCRIPTION:
E122-00-V7 (Survey 4056.03 to 4247.87)
END DESCRIPTION:
XS GIS Cut Line= 6
 3076003.745643113893212.7881513     3073290.739    13891990.662
     3072465.284    13891682.996     3072348.739    13891624.557
     3072034.984    13891595.726     3070035.877    13891412.024
#Sta/Elev= 30
  -36.02  106.27       0  102.53  634.28  104.37  753.06  101.82 1109.45  104.26
 1266.71  101.21 1438.06  103.89 1514.22  101.54 1688.33  103.91 1803.46   101.3
 1951.66  104.65 2084.36  101.72 2128.76  104.32 2347.59  102.34 2501.97  104.79
 2610.81  101.61 2791.78  104.62 2926.39  101.27  3051.9   103.7 3645.46   102.6
 4056.03  105.64 4077.75  103.57 4127.37   103.4 4166.57   90.18  4183.5   88.52
 4229.76  102.76 4265.95  104.01 4637.35  101.95 5572.69  102.92 6273.46  106.48
#Mann= 3 ,-1 , 0
  -36.02     .08       0 4077.75     .04       0 4265.95     .08       0
#XS Ineff= 2 , 0
         4054.99  105.64 4284.55           104.6
Permanent Ineff=
       F       F
Bank Sta=4127.37,4229.76
Exp/Cntr=0.3,0.1

Type RM Length L Ch R = 1 ,12779.21,1003.79,1006.01,1006.96
BEGIN DESCRIPTION:
E122-00-V8 (Survey 4016.28 to 4163.33)
END DESCRIPTION:
XS GIS Cut Line= 6
 3076039.805073113893128.1267565     3073307.567    13891948.201
     3072397.984    13891610.348      3072399.08    13891540.735
     3072404.869    13891371.711     3072435.891    13890465.851
#Sta/Elev= 30
  -10.53     106   16.38  101.95   59.55  104.12  219.13  102.29  557.49  104.48
  768.87  101.57 1145.12  104.15  1309.9  101.01 1426.56   103.9 1831.76  101.61
 1971.21  104.32 2112.62  101.79  2216.3  104.71 2530.33  104.52 2647.49  101.71
 2852.43  104.47  2952.3  101.17  3095.2   103.6 3591.89  104.47 3682.72  102.66
 4014.02  105.53 4028.28  102.88 4045.27  103.85 4085.31   89.29 4109.33   88.84
 4148.38  105.13 4166.45  104.75 4373.18  101.47 4769.74  103.78 5081.04  101.33
#Mann= 3 ,-1 , 0
  -10.53     .08       0 4014.02     .04       0 4166.45     .08       0
#XS Ineff= 2 , 0
         3974.16   105.6 4148.45          105.14
Permanent Ineff=
       F       F
Bank Sta=4045.27,4148.38
Exp/Cntr=0.3,0.1

Type RM Length L Ch R = 1 ,11773.19,998.46,1001.13,1002.61
BEGIN DESCRIPTION:
E122-00-V9 (Survey 3227.74 to 3378.01)
END DESCRIPTION:
XS GIS Cut Line= 6
 3076095.641553513893022.8577241     3073386.501    13891844.962
     3073401.647    13891581.254     3073411.487    13891409.915
     3073417.221     13891310.08     3072516.137    13890475.364
#Sta/Elev= 30
   -1.79  105.79   14.54  102.72   31.12  102.45  169.55  103.75  390.96   100.7
  699.97   103.9  792.25  101.93 1171.77  104.29 1302.01  101.14 1416.59  103.83
 1806.17   101.4 2064.19  103.79  2110.5  101.36 2288.31   104.5 2612.59  101.61
 2797.41  104.34 3051.81  102.67 3085.78  100.39 3207.15  103.13 3255.75  102.67
 3301.85   87.52 3343.95    93.5 3351.93    97.7 3356.98  102.93 3437.65  104.33
 3485.86  102.55 3894.54  100.28 4100.27  103.74 4164.74  101.27  4716.4  101.36
#Mann= 3 ,-1 , 0
   -1.79     .08       0 3207.15     .04       0 3356.98     .08       0
#XS Ineff= 2 , 0
         3208.63  103.15 3437.75          104.34
Permanent Ineff=
       F       F
Bank Sta=3255.75,3356.98
Exp/Cntr=0.3,0.1

Type RM Length L Ch R = 1 ,10772.07,997.66,995.83,994.14
BEGIN DESCRIPTION:
E122-00-V10 (Survey 2414.58 to 2563.15)
END DESCRIPTION:
XS GIS Cut Line= 6
 3076162.103207213892898.5454505     3074362.304    13892043.118
     3074390.385    13891718.507     3074413.474    13891451.592
     3074422.093    13891351.964      3072563.69    13890478.336
#Sta/Elev= 30
  -13.92   105.9    17.9  101.77    46.5  104.06  207.84   102.4  796.98  102.11
  933.75  103.49 1039.74  101.83 1224.21  104.46 1350.21   100.8 1670.84  103.96
 1928.71  103.06 2020.16   100.6 2077.89  103.57 2234.68  103.13 2296.39  100.89
 2341.55  103.43 2410.29  103.05 2421.72   101.1 2443.73  101.75 2482.93   88.29
 2493.97   87.02 2511.08   88.45  2548.2   102.8 2557.17  102.24 3619.96  101.92
 3994.43   99.93 4337.36   101.9 4512.34   99.57  4625.2   101.8 4726.07  101.53
#Mann= 3 ,-1 , 0
  -13.92     .08       0 2410.29     .04       0 2557.17     .08       0
#XS Ineff= 2 , 0
         2389.42  103.51 2548.87          102.81
Permanent Ineff=
       F       F
Bank Sta=2443.73,2548.2
Exp/Cntr=0.3,0.1

Type RM Length L Ch R = 1 ,9776.243,369.56,363.66,358.39
BEGIN DESCRIPTION:
E122-00-V11 (Survey 1658.98 to 1817.29)
END DESCRIPTION:
XS GIS Cut Line= 6
 3076210.503846813892802.1935652     3075372.087     13892402.04
     3075390.269    13891754.004      3075396.36    13891654.189
     3075412.869    13891383.615     3072584.495     13890469.42
#Sta/Elev= 30
  -26.54  105.44       0  101.97   40.07  104.51  195.11  101.58  595.47     103
  799.01  101.54  902.47  103.17  1191.1   103.4 1262.92  101.02 1307.74  102.81
 1383.12   103.1 1632.15   102.8 1664.06  100.93 1688.05  101.89 1728.15   87.52
 1744.25   86.18 1763.21   90.11 1792.28  100.89 1817.29  101.29 2143.74  102.16
 2637.98   99.61 2815.58  101.63 3001.58  100.61 3340.86  102.36 3734.32  100.37
 4106.78  101.25 4188.52   99.46 4373.06  101.01 4666.53   99.57 4894.29  101.64
#Mann= 3 ,-1 , 0
  -26.54     .08       0 1664.06     .04       0 1817.29     .08       0
#XS Ineff= 2 , 0
         1632.23   102.8 1947.27           102.4
Permanent Ineff=
       F       F
Bank Sta=1688.05,1792.28
Exp/Cntr=0.3,0.1

Type RM Length L Ch R = 1 ,9412.584,473.27,368.86,261.83
BEGIN DESCRIPTION:
E122-00-V12 (Survey 1270.27 to 1419.34)
END DESCRIPTION:
XS GIS Cut Line= 6
 3076361.360804213892540.9447878     3075780.539    13892314.704
     3075769.442    13891770.955     3075763.929    13891500.794
     3075761.888    13891400.815     3072600.129     13890458.43
#Sta/Elev= 30
   -8.86  105.38    2.83  105.07   26.57  101.27   58.19  103.61  184.22  102.93
   244.3   100.9  646.85  102.83   882.1  102.34  977.51  100.31 1025.29  102.15
 1147.95   102.9 1255.22  101.41 1278.29  100.86 1291.29  102.42 1342.28   88.72
 1362.29   85.35 1386.31   94.94 1397.49   97.11 1402.31  101.37 1902.75  101.94
 2630.74    99.7 2689.83  101.15 2964.81  100.72 3223.26  102.37 3669.23  100.43
 4006.36  101.08 4147.73    99.1 4317.76  100.34 4399.21   99.08 4827.76  101.72
#Mann= 3 ,-1 , 0
   -8.86     .08       0 1255.22     .04       0 1402.31     .08       0
#XS Ineff= 6 ,-1
  185.42 1146.58  102.91 1177.16 1290.76  102.42  1456.6 1634.77  101.39
 1666.74 1889.55  101.57 1902.66 3060.42  101.95 3129.36 4822.37  102.43
Permanent Ineff=
       F       F       F       F       F       F
Bank Sta=1291.29,1402.31
Exp/Cntr=0.3,0.1

Type RM Length L Ch R = 1 ,9043.720,224.98,226.02,227.14
BEGIN DESCRIPTION:
E122-00-V13 (Survey 813.61 to 970.77)
END DESCRIPTION:
XS GIS Cut Line= 6
  3076890.90661513891530.5605398     3076178.161    13891356.674
     3076078.244    13891352.609     3075907.483    13891345.663
     3075807.566    13891341.598     3072627.895    13890430.664
#Sta/Elev= 30
   -28.3  103.45    3.03   99.13  583.94   101.3  789.09  100.37  813.61   98.72
  821.61  100.44  843.63   98.77  872.73   87.93  875.68   85.81  881.76   84.95
  885.76   85.62  886.76   87.21  895.71    88.3  930.76  101.31  964.44  101.98
  998.29   103.1 1041.87  100.81 1468.82  101.45 1929.63    99.3 2033.62  100.87
 2119.93   99.56 2368.32   99.99 2415.13  101.55 2466.86  100.76 2709.28  102.41
 2942.33   99.84 3491.77   99.62 3564.22  100.61 3740.63   98.62 4383.84  101.86
#Mann= 3 ,-1 , 0
   -28.3     .08       0  789.09     .04       0  964.44     .08       0
#XS Ineff= 2 , 0
          584.15  101.31  998.52          103.11
Permanent Ineff=
       F       F
Bank Sta=821.61,930.76
Exp/Cntr=0.3,0.1

Type RM Length L Ch R = 1 ,8817.703,55.01,66.39,80.7
BEGIN DESCRIPTION:
E122-00-SV9 (Survey 936.32 to 1055.41) XS 4
END DESCRIPTION:
XS GIS Cut Line= 6
 3077025.522869413891269.3030915     3076360.297    13891144.145
     3076193.703    13891134.421     3075732.261    13891107.489
      3073356.78     13890607.74     3072667.481    13890386.811
#Sta/Elev= 30
  -22.51  103.35       0  101.94  130.18  101.24  160.71   99.32   415.2  100.08
  439.56   98.94  465.97  100.41  709.31   99.85  769.41  101.09  931.31   99.76
  936.32   99.53 1007.38   85.43 1055.41  100.65 1153.05  101.79 1749.12   97.81
 2263.68  100.46 2382.02   98.78 2554.55   99.03 2651.86   101.3 2717.04   99.64
 2920.35  101.26 3042.98   98.33 3273.94  100.38 3573.96   98.58 3632.97  100.26
 3733.36   98.49 3773.71   99.98 3980.31  100.28 4076.45   102.5 4434.81   102.1
#Mann= 3 ,-1 , 0
  -22.51     .08       0  931.31     .04       0 1153.05     .08       0
#XS Ineff= 2 , 0
          768.39  101.11  1205.2          102.37
Permanent Ineff=
       F       F
Bank Sta=936.32,1055.41
Exp/Cntr=0.5,0.3

Type RM Length L Ch R = 1 ,8751.316,45.44,44.36,43.04
BEGIN DESCRIPTION:
E122-00-S9 (Survey 977.93 to 1068.79) XS 3
END DESCRIPTION:
XS GIS Cut Line= 6
 3077025.627359513891249.6226134     3076174.831    13891091.838
        3075819.    13891025.848     3075243.629    13890934.322
     3073392.835    13890600.082     3072669.478    13890360.626
#Sta/Elev= 30
  -13.22  103.64   17.46     101   139.5  101.53  169.23   99.61  574.64  100.55
  932.25   98.48  954.58   99.08  977.93   97.04 1018.97   85.57 1068.79   99.18
 1154.21   99.94 1344.13  100.22 1386.12   96.85 1450.45   95.93 1708.66   98.02
 1768.87   96.21 2039.13   98.29 2541.69   97.48 2653.39   100.2 2699.12   98.06
 2805.82   98.22 2897.27  100.97  3049.7   97.76 3293.58  100.18 3339.31   98.61
 3569.24    98.2 3631.14   99.97 3719.78   98.29 4032.69  102.45 4439.28   101.9
#Mann= 3 ,-1 , 0
  -13.22     .08       0  932.25     .04       0 1154.21     .08       0
#XS Ineff= 2 , 0
          953.37   99.08 1223.84          101.16
Permanent Ineff=
       F       F
Bank Sta=954.58,1068.79
Exp/Cntr=0.5,0.3

Type RM Length L Ch R = 3 ,8747.55 ,,,
BEGIN DESCRIPTION:
Structure 9 - Breen Road
END DESCRIPTION:
Bridge Culvert--1,0,-1,-1, 0
Deck Dist Width WeirC Skew NumUp NumDn MinLoCord MaxHiCord MaxSubmerge Is_Ogee
3.76,37.1,2.6,0, 61, 62, 100.6792, , 0.95, 0, 0,0,,
       0   52.86  178.11  188.99  207.53   916.9  971.98 1028.86    1092  1157.1
 1347.95  1398.3 1400.49 1441.54 1476.68 1479.87 1610.42 1724.86 1991.64 2017.15
 2132.61 2140.27 2165.99 2226.68 2272.28 2288.84 2317.82 2342.42 2363.08  2483.6
 2511.02 2604.36 2624.42 2634.14 2648.71 2785.42 2810.96 2842.86 2935.25 2954.77
 2988.53  3001.6 3015.56 3056.27 3098.16 3111.53  3136.8    3178 3221.29 3287.04
 3367.54 3386.21 3462.69 3481.78 3525.78 3580.61 3653.07 3691.12  3886.5 3930.95
 4155.81
     103     102     101     101     101   100.9  100.68  100.75  100.71  100.73
     100      99      99      99      99      99      98      97      97      97
      97      97      97      97      97      97      97      97      97      97
      97      98      99      99      98      98      99     100     100      99
      98      98      98      98      98      98      98      98      99      99
      99      99      99      99      99      99      99     100     101     102
     102
                                           98.45   98.45   98.45   98.45   98.45
                                                                                
                                                                                
                                                                                
                                                                                
                                                                                
        
     -25   19.13   71.99  197.24  208.12  226.66  936.03  991.11 1047.99 1111.13
 1176.23 1367.08 1417.43 1419.62 1460.67 1495.81    1499 1629.55 1743.99 2010.77
 2036.28 2151.74  2159.4 2185.12 2245.81 2291.41 2307.97 2336.95 2361.55 2382.21
 2502.73 2530.15 2623.49 2643.55 2653.27 2667.84 2804.55 2830.09 2861.99 2954.38
  2973.9 3007.66 3020.73 3034.69  3075.4 3117.29 3130.66 3155.93 3197.13 3240.42
 3306.17 3386.67 3405.34 3481.82 3500.91 3544.91 3599.74  3672.2 3710.25 3905.63
 3950.08 4174.94
     103     103     102     101     101     101     101     101     101     101
     101     100      99      99      99      99      99      98      97      97
      97      97      97      97      97      97      97      97      97      97
      97      97      98      99      99      98      98      99     100     100
      99      98      98      98      98      98      98      98      98      99
      99      99      99      99      99      99      99      99     100     101
     102     102
                                                   98.45   98.45   98.45   98.45
   98.45
                                                                                
                                                                                
                                                                                
                                                                                
                
Pier Skew, UpSta & Num, DnSta & Num=  ,1016.5, 4 ,1016.5, 4 , 3 , 3 , 0 ,,
    1.35    1.35       2       2
 85.5686   95.95   95.95   98.45
    1.35    1.35       2       2
   85.25   95.95   95.95   98.45
Pier Skew, UpSta & Num, DnSta & Num=  ,1058.77, 4 ,1058.77, 4 , 3 , 3 , 0 ,,
    1.35    1.35       2       2
 85.5686  95.957  95.957  98.457
    1.35    1.35       2       2
 85.2476  95.957  95.957  98.457
BR Coef=-1 , 1 , 1 ,1.25, 0 ,,,0.8,-1,2,0,
WSPro=,,,, 1 ,,,, 0 ,,,, 0 ,,,,-1 ,-1 ,-1 , 0 , 0 , 0 , 0 , 0
BC Design=,, 0 ,, 0 ,,,,,,
BC HTab HWMax=103.64

Type RM Length L Ch R = 1 ,8706.955,77.64,76.18,75.28
BEGIN DESCRIPTION:
Survey 1029.4 to 1038.1 from S9 XS 2
END DESCRIPTION:
XS GIS Cut Line= 6
 3077065.0352328 13891194.709689     3076178.491    13891044.679
     3076079.893    13891027.994      3075935.29    13891003.522
     3075836.691    13890986.836     3072729.342    13890300.762
#Sta/Elev= 30
  -24.45     103     .47     100   23.33   99.43  503.82   99.14  592.13  100.33
  654.43    99.4  715.49  100.18  924.74   99.53  989.33  100.01 1004.55   97.76
 1019.76   92.66  1029.4    86.6  1038.1   85.44 1095.83   98.44 1120.14   99.95
 1321.06  100.04  2092.5   99.18 2132.64   98.39 2277.42  100.59 2896.67   99.33
 3138.55  100.31  3170.1  101.91 3342.88  100.79 3435.02  101.78 3576.11  100.94
 3743.27  102.31 3798.19  101.22 3815.43  102.35  3944.6  102.54 4403.55   101.5
#Mann= 5 ,-1 , 0
  -24.45     .08       0  924.74     .06       0  989.33     .08       0
 1120.14     .06       0 1321.06     .08       0
#XS Ineff= 2 , 0
          988.65  100.09 1242.79          100.62
Permanent Ineff=
       F       F
Bank Sta=989.33,1120.14
Exp/Cntr=0.5,0.3

Type RM Length L Ch R = 1 ,8630.772,535.79,540.54,529.77
BEGIN DESCRIPTION:
Survey 1084.66 to 1093.42 (1029.4 to 1038.1 from S9) XS 1
END DESCRIPTION:
XS GIS Cut Line= 6
 3077115.487725313891100.8101042     3076191.077    13890965.704
     3076092.128    13890951.243     3075947.525    13890930.108
     3075848.576    13890915.647     3072764.263    13890250.875
#Sta/Elev= 30
  -21.81  102.82    8.38   98.56   79.92  100.23  360.52   99.62  539.11  101.28
  698.72   99.86  971.01  101.21 1015.15  100.86 1036.09  100.14 1084.66   86.37
 1093.42   85.21 1145.34   99.36 1147.56   99.49 1216.19  101.47 1368.25  101.28
 1438.74   99.79 1483.46  100.89 1558.91   99.39 1967.08   98.18 2129.25    98.7
 2307.19  101.38 2410.77   99.99 3078.28   99.47 3172.36   101.5 3479.46  102.55
  3629.9  101.34 3775.45  102.88 3852.44  101.08 3940.68  102.52  4413.7  102.01
#Mann= 5 ,-1 , 0
  -21.81     .08       0  971.01     .06       0 1015.15     .08       0
 1147.56     .06       0 1368.25     .08       0
#XS Ineff= 2 , 0
           991.2   101.7 1297.36          101.91
Permanent Ineff=
       F       F
Bank Sta=1036.09,1145.34
Exp/Cntr=0.3,0.1

Type RM Length L Ch R = 1 ,8090.234,725.17,723.56,711.4
BEGIN DESCRIPTION:
E122-00-V14 (Survey 1227.14 to 1394.35)
END DESCRIPTION:
XS GIS Cut Line= 6
  3077403.22419513890567.1258819     3076174.911    13890423.557
     3075996.626    13890402.718     3075897.302    13890391.109
     3075492.508    13890343.795     3072983.764    13890036.362
#Sta/Elev= 30
  -21.12  101.66    6.13   98.32  628.52   99.83  687.47    98.7  736.76   100.6
  766.97   99.11 1099.42   99.19 1196.13  101.62  1240.4   99.38 1292.94   88.35
 1300.89   85.38 1301.99   83.65  1308.3   83.59  1310.4   86.97 1344.76   92.59
 1354.92  100.33 1362.98   97.61 1373.34   97.84 1388.39   98.16 1394.35  100.06
 1567.38  100.66 1722.18   98.38 2569.36   98.19 3418.57  103.24 3529.77  101.87
 3564.45   104.2 3744.66  101.49 3836.26   102.6 4002.66  100.69 4430.11  101.05
#Mann= 5 ,-1 , 0
  -21.12     .08       0 1196.13     .06       0  1240.4     .08       0
 1373.34     .06       0 1567.38     .08       0
#XS Ineff= 3 ,-1
  -21.12 1189.71  101.79    1355 1472.41  100.33 1567.14 3076.19  100.67
Permanent Ineff=
       F       F       F
Bank Sta=1240.4,1354.92
Exp/Cntr=0.3,0.1

Type RM Length L Ch R = 1 ,7366.673,43.95,43.51,43.3
BEGIN DESCRIPTION:
E122-00-SV10 (Survey 1682.58 to 1754.59) XS 4
END DESCRIPTION:
XS GIS Cut Line= 6
     3077818.016    13889738.712     3076283.563     13889700.19
     3076045.249    13889694.207     3075945.281    13889691.697
     3075478.096    13889682.167     3073043.628    13889946.567
#Sta/Elev= 30
       0      98  333.13   98.83  996.89   97.04  1195.6   98.32  1580.5   97.47
 1623.67   97.95 1652.34   95.83 1682.58   86.47  1697.1   85.36 1700.13   82.47
 1703.28   82.03  1713.1   86.08 1727.59   89.03 1741.61   96.43 1772.07   96.65
 1783.11   97.48 1963.65   96.63 2085.15   96.36 2450.32   99.59 2663.84   99.34
 2784.17   101.5 2870.88   99.84 2974.53  101.42 3112.43  100.94 3169.72   99.63
 3326.13  101.43 3777.31  101.18 4030.26  102.67 4272.48  101.43 4789.39  101.13
#Mann= 5 ,-1 , 0
       0     .08       0  1580.5     .06       0 1652.34     .08       0
 1772.07     .06       0 1963.65     .08       0
#XS Ineff= 3 ,-1
  684.11 1193.81   98.31 1284.83 1605.22   98.01 1783.62 2235.08   97.48
Permanent Ineff=
       F       F       F
#Block Obstruct= 2 , 0
          183.81   98.83
Bank Sta=1652.34,1741.61
Exp/Cntr=0.5,0.3

Type RM Length L Ch R = 1 ,7323.165,54.41,54.35,54.3
BEGIN DESCRIPTION:
E122-00-S10 (Survey 1720.64 to 1785.49) XS 3
Data inserted from bridge survey
END DESCRIPTION:
XS GIS Cut Line= 6
     3077849.309    13889685.976     3076178.385    13889653.688
     3076058.563    13889651.372     3075958.582     13889649.44
     3075476.232    13889666.352     3073078.549    13889916.635
#Sta/Elev= 30
       0   98.51   18.47   97.83  183.15   98.67  721.08   98.47  998.97   96.69
 1242.33   98.15 1626.71   97.05 1720.64   96.83 1720.73    80.1 1744.23   80.13
 1744.64   96.82 1772.51   96.43 1814.18   97.34 1961.62    96.7  2001.2   95.88
 2236.33   97.15 2494.21   99.83 2687.11   99.65 2817.59  101.19 2898.14   99.92
 3027.96  101.21 3186.55   99.69 3440.38  101.81 3591.07  101.21 3749.77  101.93
 3816.16  101.11 4237.23  102.97 4388.62  101.41 4540.49  102.28 4784.44  101.85
#Mann= 5 ,-1 , 0
       0     .08       0 1626.71     .06       0 1720.64     .08       0
 1772.51     .06       0 1961.62     .08       0
#XS Ineff= 4 ,-1
  735.76 1241.82   98.14 1443.43 1657.37   97.45 1744.79 1800.01   96.82
 1814.49 2246.79   97.34
Permanent Ineff=
       F       F       F       F
#Block Obstruct= 2 , 0
          213.32   98.68
Bank Sta=1720.64,1744.64
Exp/Cntr=0.5,0.3

Type RM Length L Ch R = 2 ,7296.664,,,
BEGIN DESCRIPTION:
Structure 10
END DESCRIPTION:
Bridge Culvert--1,0,-1,-1, 0
Deck Dist Width WeirC Skew NumUp NumDn MinLoCord MaxHiCord MaxSubmerge Is_Ogee
0.5,50,2.6,0, 6, 6, 96, , 0.95, 0, 0,0,,
 1651.12 1720.53 1720.53 1744.52 1744.52 1783.12
   96.77      96    96.9    96.9      96   96.45
      75      75      75      75      75      75
 1676.25 1745.66 1745.66 1769.65 1769.65 1808.25
   96.77      96    96.9    96.9      96   96.45
      75      75      75      75      75      75
BR Coef=-1 , 0 , 0 ,, 0 ,,,0.8,-1,,1,
WSPro=,,,, 1 ,,,, 0 ,,,, 0 ,,,,-1 ,-1 ,-1 , 0 , 0 , 0 , 0 , 0
Multiple Barrel Culv=2,9.1,11,50,0.013,0.4,1,8,1,80.1,80.4, 2,Culvert #1  , 0 ,0.5
 1726.63 1751.76 1738.43 1763.56
Culvert Bottom n=0.013
BC Design=,, 0 ,, 0 ,,,,,,
BC HTab HWMax=102.97

Type RM Length L Ch R = 1 ,7268.812,19.6,19.01,18.45
BEGIN DESCRIPTION:
Survey 1745.38 to 1810.23 XS 2
Data inserted from bridge survey
END DESCRIPTION:
XS GIS Cut Line= 6
     3077875.405    13889632.118       3076179.8    13889599.353
     3076059.978    13889597.038     3075959.996    13889595.106
     3075343.483    13889583.192     3073198.277    13889786.929
#Sta/Elev= 30
       0   98.05  754.97   98.23 1146.33   96.65 1285.55   97.95 1540.23   96.39
 1640.54   96.68 1745.38   96.83 1745.47   80.42 1768.97   80.39 1769.38   96.82
 1828.03   97.06 1968.65    96.5 1998.67   95.81 2161.83   97.53 2218.18   97.19
 2445.93    98.5 2598.05  100.92 2719.97  100.93 2867.65   98.87 3027.63  100.49
 3423.42  102.09 3576.69  102.08 3660.47  100.92 3931.68  102.06 3961.82  101.23
 4013.54  102.05 4070.43  101.39 4411.19  101.69 4539.35  103.25 4687.25  102.93
#Mann= 5 ,-1 , 0
       0     .08       0 1640.54     .06       0 1745.38     .08       0
 1828.03     .06       0 1968.65     .08       0
#XS Ineff= 5 ,-1
  769.02 1279.62   97.95 1488.29 1688.09   96.89 1769.17 1810.59   96.82
 1850.27 2154.71   97.45 2162.25 2277.99   97.54
Permanent Ineff=
       F       F       F       F       F
#Block Obstruct= 2 , 0
          166.29    98.5
Bank Sta=1745.38,1769.38
Exp/Cntr=0.5,0.3

Type RM Length L Ch R = 1 ,7249.799,345.63,350.98,346.3
BEGIN DESCRIPTION:
Survey 1777.29 to 1790.34  XS 1
END DESCRIPTION:
XS GIS Cut Line= 6
     3077898.837    13889594.237     3076287.785    13889580.584
     3076056.534    13889578.625     3075956.537    13889577.777
     3075278.469    13889572.031     3073243.175     13889747.02
#Sta/Elev= 30
       0   98.19  782.56    98.1 1186.79   96.64  1310.8   97.83 1709.95   96.78
 1725.41   96.18 1728.43   96.04 1770.93   87.95 1773.44   87.19 1777.29   82.47
 1780.31   82.03 1790.34   86.08 1812.37   90.87 1819.22   93.53 1828.34   95.25
 1848.44   96.68 1883.52   97.35  2005.2   96.15 2058.45   95.71  2472.3    98.5
 2636.83  100.94 2767.21  100.98 2920.35    98.8 3353.97  102.01 3607.27  102.01
 3682.37  100.96  4002.2  101.96 4160.61  100.75 4287.28  102.58 4663.27  103.06
#Mann= 5 ,-1 , 0
       0     .08       0 1709.95     .06       0 1725.41     .08       0
 1848.44     .06       0  2005.2     .08       0
#XS Ineff= 4 ,-1
  207.79  522.94   98.38  824.23 1309.07   97.84 1883.63 2145.53   97.33
 2164.24 2295.19   97.53
Permanent Ineff=
       F       F       F       F
#Block Obstruct= 2 , 0
          204.33   98.53
Bank Sta=1728.43,1848.44
Exp/Cntr=0.3,0.1

Type RM Length L Ch R = 1 ,6898.815,909.08,915.81,914.45
BEGIN DESCRIPTION:
E122-00-V15 (Survey 1827.7 to 1979.81)
END DESCRIPTION:
XS GIS Cut Line= 6
     3078060.878    13889291.733     3076340.856    13889240.474
       3076240.9    13889237.495     3076066.088    13889232.286
     3075966.132    13889229.307     3073786.909    13889164.363
#Sta/Elev= 30
       0   98.12 1161.77   97.27 1498.46   96.07 1596.19   94.92 1795.86   95.83
  1827.7   95.12 1865.74   95.59 1881.38   87.66 1892.73   87.23 1904.57    81.3
 1908.57   80.97  1915.6   86.93 1929.83   88.09 1949.85   96.04 2011.31   97.47
 2399.98   98.34 2545.71   98.06 2881.45  100.28 3016.75  100.06 3046.76    99.1
 3099.11  100.66 3184.67   99.96 3448.88  101.06 3489.33  100.17 3640.48  100.98
 3855.07   99.99 3922.46   101.4 4148.67  102.51 4241.62  102.03 4275.87  100.73
#Mann= 5 ,-1 , 0
       0     .08       0 1795.86     .06       0 1865.74     .08       0
 1949.85     .06       0 2399.98     .08       0
#XS Ineff= 3 ,-1
  422.92  779.06   97.88 1509.97 1807.68   95.98 1818.81 1863.33    95.6
Permanent Ineff=
       F       F       F
#Block Obstruct= 2 , 0
           72.34   98.16
Bank Sta=1865.74,1949.85
Exp/Cntr=0.3,0.1

Type RM Length L Ch R = 1 ,5983.005,554.169,551.039,542.586
BEGIN DESCRIPTION:
E122-00-V16 (Survey 2233.55 to 2404.95)
END DESCRIPTION:
XS GIS Cut Line= 6
      3078492.13    13888483.559     3076375.392    13888336.778
     3076275.631     13888329.86     3076117.027    13888318.862
     3076017.266    13888311.944     3074657.313    13888217.641
#Sta/Elev= 30
       0   95.53  516.87   96.78  646.09   96.57  691.32   95.74  789.09   96.35
  852.63   95.11  887.21   95.54  995.37   94.64 1105.81   94.61 1215.93   95.94
  2191.1   93.89 2233.55   93.87 2265.55   94.71 2281.65   86.56 2295.68    85.3
 2300.81   81.41 2301.74   80.15 2306.52   79.25  2311.5   81.58 2316.42   85.22
 2331.23   86.62 2347.31   95.01 2404.95   96.35 2523.83   96.15 2608.26   97.43
 3028.49   98.94 3421.18   98.12 3502.44   97.93  3541.6   98.76 3844.03   98.03
#Mann= 5 ,-1 , 0
       0     .08       0  2191.1     .06       0 2265.55     .08       0
 2347.31     .06       0 3421.18     .08       0
#XS Ineff= 2 , 0
         2264.23   94.72 3123.52           99.14
Permanent Ineff=
       F       F
Bank Sta=2265.55,2347.31
Exp/Cntr=0.5,0.3

Type RM Length L Ch R = 1 ,5431.968,80.601,83.961,79.494
BEGIN DESCRIPTION:
E122-00-V16 (Survey 2233.55 to 2404.95 copied from section 5983. Elevations of survey data adjusted to fit stream slope).
END DESCRIPTION:
XS GIS Cut Line= 6
     3078656.303    13887845.789     3076534.784    13887809.991
     3076434.798    13887808.304     3076275.836    13887805.621
      3076175.85    13887803.934     3074812.825    13887780.935
#Sta/Elev= 30
       0   94.02  109.76   94.17  182.23   92.09  212.24   93.76  272.14    94.2
 1293.61    93.6 1393.28   92.48 1592.43   94.11 1967.49   93.49  2072.8   92.88
 2117.51    91.1 2229.54   93.29 2267.87   93.61 2267.98   92.51 2271.82   89.95
 2275.98   85.46 2283.95    84.2 2304.01   78.17 2308.78   78.15 2318.68   84.12
 2341.36   93.91 2407.08   96.35 2426.01   93.93 2525.95    93.6  2747.6   95.26
 2837.61   94.92 2964.81   96.61  3536.5   96.94 3629.58   96.36 3844.03   97.61
#Mann= 5 ,-1 , 0
       0     .08       0 2229.54     .06       0 2267.87     .08       0
 2341.36     .06       0  3536.5     .08       0
#XS Ineff= 2 , 0
         2268.02   93.65 2406.51           96.39
Permanent Ineff=
       F       F
Bank Sta=2267.87,2341.36
Exp/Cntr=0.5,0.3

Type RM Length L Ch R = 5 ,5380    ,,,
BEGIN DESCRIPTION:
Inline weir, structure 11 - Shape taken from survey of structure
END DESCRIPTION:
IW Pilot Flow=0
#Inline Weir SE= 18
    2272  88.259 2286.02  88.393 2287.02  86.425 2292.01  86.461 2293.01  84.587
 2297.03  84.517 2297.03  82.727 2301.01  82.805 2302.03  81.388 2302.03  78.836
 2307.01  81.218 2307.01  82.728 2312.03  82.713 2312.03  84.245 2316.03  84.275
 2322.03  85.599 2323.03  88.034    2335  88.034
IW Dist,WD,Coef,Skew,MaxSub,Min_El,Is_Ogee,SpillHt,DesHd
45,1,2.6,0,0.95,, 0 ,,,0,0,

Type RM Length L Ch R = 1 ,5348.006,80.34,80.35,78.43
BEGIN DESCRIPTION:
E122-00-S11 (Survey 2403.54 to 2499.54)
END DESCRIPTION:
XS GIS Cut Line= 6
     3078795.461    13887746.543     3076516.288    13887728.088
     3076416.291    13887727.279     3076273.316    13887726.121
     3076173.319    13887725.311     3075124.561    13887716.819
#Sta/Elev= 30
       0   92.65  137.17   93.03   202.1   94.01  243.92   93.77  285.01   91.09
  615.02   93.08   903.8    92.2  1350.8   93.25 1484.49   92.84 1536.23   91.31
    1569   93.05 1676.43   93.72 2071.76   93.21 2152.44   92.43  2322.5   93.11
 2349.45   92.49 2403.54   91.44 2421.53    80.6 2433.53   76.92 2460.54   76.03
 2499.54   92.77    2533   92.86 2602.57   93.63 2673.24   92.18 2730.09   94.08
 3039.97   96.52 3343.74   96.98 3362.62   96.16 3472.76   96.23 3671.02   96.95
#Mann= 5 ,-1 , 0
       0     .08       0 2349.45     .04       0 2403.54    .015       0
 2499.54     .04       0    2533     .08       0
#XS Ineff= 2 , 0
         1820.88   93.84 2588.24           93.69
Permanent Ineff=
       F       F
Bank Sta=2403.54,2499.54
Exp/Cntr=0.5,0.3

Type RM Length L Ch R = 1 ,5267.653,503.58,505.14,506.35
BEGIN DESCRIPTION:
E122-00-SV11 (Survey 2397.82 to 2513.91)
END DESCRIPTION:
XS GIS Cut Line= 6
      3078791.84    13887628.789     3076520.919    13887646.058
     3076420.922    13887646.819     3076268.685    13887647.976
     3076168.688    13887648.737     3075146.468     13887656.51
#Sta/Elev= 30
       0   92.54  130.99   92.95  155.79   93.89  711.43   93.57   866.4   92.84
  904.56   91.34 1166.21   92.91 1671.18   92.48 1946.43   91.96 2182.38   89.58
 2295.59   92.51 2369.56   90.63 2397.92   90.56 2415.91    83.4 2431.91   79.47
  2438.9   75.31 2443.91   75.16 2451.88    75.4  2456.9   80.22 2471.91   83.78
 2492.92   92.46 2515.38   92.16 2546.45   93.32 2605.98   93.46 2686.96   91.99
 2710.07   93.05 2876.46   94.54 3300.76   97.14 3356.47   96.15 3645.48   96.62
#Mann= 3 ,-1 , 0
       0     .08       0 2369.56     .04       0 2515.38     .08       0
#XS Ineff= 3 ,-1
       0 2295.02   92.53 2492.84 2523.59   92.46 2605.18 3645.48   93.48
Permanent Ineff=
       F       F       F
Bank Sta=2397.92,2492.92
Exp/Cntr=0.3,0.1
